HEC-RAS study MILLERRN.prj: MILLERRN

--- MILLERRN.g01 (geometry) --- (continued)

Type RM Length L Ch R = 1 ,10086   ,259.2,247.2,224.1
XS GIS Cut Line= 2
2470653.06611135580724.1057923272471277.37640033580615.841726857
#Sta/Elev= 30
       0 1823.12    46.4 1801.21    99.1 1778.25   109.8 1772.12   123.5 1762.38
   131.6 1758.85   139.7 1757.77   151.9 1757.72   168.2 1758.48   180.3 1760.08
   257.5 1761.61   273.7  1759.8   289.9 1761.03     310 1757.69   341.6 1756.15
   355.4 1758.05   371.1 1759.17   399.6 1758.58   410.8 1761.95   415.8 1762.21
   431.5 1761.49   452.3 1758.69   464.5 1759.66   517.3 1759.25   529.5 1760.11
   549.8 1756.99   553.8 1758.26     566 1767.29   574.1 1770.94   633.6 1785.48
#Mann= 7 ,-1 , 0
       0      .1       0   93.84      .1       0  292.48      .1       0
     310    .045       0   355.4      .1       0   391.8     .06       0
  491.13      .1       0
#XS Ineff= 2 , 0
          289.21 1769.71  413.86         1768.09
Permanent Ineff=
       F       F
Bank Sta=310,355.4
XS Rating Curve= 0 ,0
Exp/Cntr=0.3,0.1

Type RM Length L Ch R = 1 ,9839    ,102.2,97.5,89.4
XS GIS Cut Line= 3
2470712.68627042 581013.282142832470964.38453648580989.233719173
2471238.97368315580664.501937212
#Sta/Elev= 30
       0 1787.21    22.2 1779.89    38.2 1776.41    74.4 1773.12   102.5 1769.47
   114.6 1764.78   130.7 1756.14   134.7 1754.86   162.8 1755.42   198.5 1752.32
   219.1 1754.43   231.1 1753.56   268.9 1754.87   304.4 1754.43     345 1756.46
   360.7 1753.92   378.2 1755.92   388.4 1752.18   407.8 1751.16   426.5 1752.64
     435 1755.76   503.1 1753.71   554.2 1758.28   597.2  1757.8   615.8 1756.51
   640.6 1757.53     645 1758.95   653.5 1764.79   664.5 1770.75   678.1 1776.89
#Mann= 7 ,-1 , 0
       0      .1       0  147.36     .12       0   262.3      .1       0
  289.17     .12       0   388.4    .045       0   426.5     .06       0
  550.67      .1       0
#XS Ineff= 2 , 0
          377.02  1760.1  436.58         1760.26
Permanent Ineff=
       F       F
Bank Sta=388.4,426.5
XS Rating Curve= 0 ,0
Exp/Cntr=0.5,0.3

Type RM Length L Ch R = 1 ,9741    ,95.8,75.9,75.6
XS GIS Cut Line= 3
2470682.26433993581084.5943399272471091.40136493 581040.83619353
2471242.32017243580675.263103693
#Sta/Elev= 30
       0 1771.82   121.2 1764.38   133.8 1762.09   165.4 1753.08   177.5 1752.33
   257.9 1754.01   278.2 1749.81   302.2 1749.73   322.3 1752.94   346.4 1750.69
   370.6 1753.07   430.7 1753.41   448.2 1752.53   500.1 1753.55   509.6 1750.78
   514.6 1748.81   521.8 1748.27     535 1748.89   541.1 1750.68   556.4 1755.55
   569.4 1753.44   582.3  1753.6   595.3 1756.13   620.7 1756.54     630 1754.53
   707.8 1755.37   772.8 1757.97     777 1759.11   789.2 1769.53     807 1776.98
#Mann= 5 ,-1 , 0
       0     .12       0   430.7     .06       0   509.6    .045       0
   541.1     .06       0   620.7      .1       0
#XS Ineff= 2 , 0
          485.09  1755.4  554.39          1755.6
Permanent Ineff=
       F       F
Bank Sta=509.6,541.1
XS Rating Curve= 0 ,0
Exp/Cntr=0.5,0.3

Type RM Length L Ch R = 1 ,9665    ,63.1,106,129.9
XS GIS Cut Line= 3
2470710.31513201581121.9679742132471138.88200314581083.877764217
2471319.10912194 580710.66009003
#Sta/Elev= 30
       0 1767.72    36.6 1764.71    85.2    1756   124.9  1751.5   182.2 1753.59
   261.5 1753.53   273.5 1750.68   290.9 1748.97   337.8 1752.14   418.1 1753.14
   435.8 1751.54   453.6 1752.67   475.9 1751.95   487.8 1750.13   512.7 1747.68
   540.3 1748.08   547.7 1749.74   560.2 1755.44   600.1 1754.84   693.4 1760.81
   720.1 1757.92   742.3 1760.99   760.1 1753.98   764.5 1754.29   786.7 1759.11
   808.9  1760.5   816.3 1762.28   822.2 1765.11   835.3 1775.68   844.7 1779.77
#Mann= 6 ,-1 , 0
       0      .1       0  200.84     .12       0  399.99     .06       0
   487.8    .045       0   547.7     .06       0  550.82      .1       0
#XS Ineff= 2 , 0
          418.42 1757.12  558.77         1757.62
Permanent Ineff=
       F       F
Bank Sta=487.8,547.7
XS Rating Curve= 0 ,0
Exp/Cntr=0.5,0.3

Type RM Length L Ch R = 1 ,9559    ,259.5,269.4,274.3
XS GIS Cut Line= 2
2470673.58070916581162.2318546482471316.47425757581086.149777914
#Sta/Elev= 30
       0 1767.74    33.4 1765.98    53.5  1763.5    65.6 1761.01    88.9 1753.99
      98 1752.66     130 1752.84   154.2 1750.65   178.4 1751.96   226.7 1751.45
   238.8 1752.79     259 1753.18   275.1 1750.53   295.2 1751.48   326.5 1748.57
   355.6 1752.16   395.9 1752.33     408 1751.32   452.3 1753.03   472.3 1751.89
   486.7 1748.66   496.6  1746.3   508.3 1746.13   512.7 1746.47   516.7 1748.22
   528.8 1757.64   533.5 1760.55   585.2 1786.87   617.4 1801.47   647.4 1812.82
#Mann= 6 ,-1 , 0
       0      .1       0  243.24     .12       0  442.06     .06       0
   486.7    .045       0   516.7     .06       0  541.47     .12       0
#XS Ineff= 2 , 0
           450.7 1759.55
Permanent Ineff=
       F       F
Bank Sta=486.7,516.7
XS Rating Curve= 0 ,0
Exp/Cntr(USF)=0,0
Exp/Cntr=0.3,0.1

Type RM Length L Ch R = 1 ,9290    ,199.3,197.4,191.4
XS GIS Cut Line= 2
 2470650.3895809581242.3129691432471278.03087478581402.074623565
#Sta/Elev= 30
       0 1765.66      51  1761.9    58.2 1760.09    74.7 1752.61    82.9 1750.51
   107.7 1750.73   124.2 1748.48   165.5 1747.18     215    1747   239.8 1749.38
   256.3  1748.9   264.5  1746.3   272.8 1745.39   326.7  1746.6   351.2 1748.59
     389 1747.91   413.1 1749.69   425.2 1749.05   431.8 1744.87   437.9 1742.72
   446.1 1741.95   458.1 1742.32   466.8  1744.8   487.4 1753.91   499.8 1764.55
   512.2 1771.73   525.7 1777.46   536.9 1781.12   558.9 1784.75   647.7 1793.78
#Mann= 7 ,-1 , 0
       0      .1       0  195.63     .12       0  215.28      .1       0
  303.92     .06       0   431.8    .045       0   466.8      .1       0
   520.5     .12       0
#XS Ineff= 2 , 0
          419.22 1758.83
Permanent Ineff=
       F       F
Bank Sta=431.8,466.8
XS Rating Curve= 0 ,0
Exp/Cntr=0.3,0.1

Type RM Length L Ch R = 1 ,9093    ,200.8,216.1,230.7
XS GIS Cut Line= 3
2470530.26816463581390.1081428582470842.33540136581530.776503401
2471318.33134422581558.044468027
#Sta/Elev= 30
       0 1779.12    70.5 1765.46    76.6 1763.13    97.1  1752.9   114.6 1748.71
   127.8 1747.34   276.2 1745.51   288.3 1744.84   307.7  1742.4   325.2 1744.84
   342.6 1745.66   406.8 1744.16   442.9 1740.86     535 1746.25   551.1 1745.34
   559.4 1743.03   567.1 1740.12   583.1 1739.66   591.1 1740.32   597.6 1742.58
   603.1 1743.42   611.2 1743.38   619.2 1745.16   623.2 1746.77   647.2 1761.16
   659.2 1767.25   679.3  1775.5   687.3 1777.72   784.6 1792.56   819.1 1795.62
#Mann= 7 ,-1 , 0
       0      .1       0  266.53     .12       0  379.29      .1       0
  481.02     .06       0   559.4    .045       0   597.6     .12       0
  684.46      .1       0
#XS Ineff= 2 , 0
           538.6 1750.67
Permanent Ineff=
       F       F
Bank Sta=559.4,597.6
XS Rating Curve= 0 ,0
Exp/Cntr=0.5,0.3

Type RM Length L Ch R = 1 ,8876    ,62.9,64.6,67.2
XS GIS Cut Line= 4
2470526.94919265581451.6070888172471017.98435304581642.815844066
2471222.13792561581900.2268703492471390.08571184582010.958918693
#Sta/Elev= 30
       0 1778.21    42.7 1766.93    73.4  1750.9   111.4 1746.11   270.2 1744.67
   295.9 1741.88   326.8 1745.15   373.2 1744.56   403.3 1741.78   447.3  1740.5
   573.2 1742.65   637.6 1741.47   647.1 1738.97   661.4 1736.03   669.8 1736.34
   676.2 1738.47   695.4 1746.29   734.2 1754.38   751.7  1755.1     761 1756.98
     767  1756.3   787.4 1747.14     805 1755.93     818 1760.42   856.2 1771.31
   866.5 1770.49   878.1 1771.59   889.6 1779.22   918.5 1788.75  1056.7  1828.5
#Mann= 10 ,-1 , 0
       0      .1       0  182.78     .12       0  377.24      .1       0
  388.46     .12       0  503.71     .06       0  552.76    .055       0
   647.1    .045       0   676.2     .06       0  880.33      .1       0
 1015.27     .12       0
#XS Ineff= 3 ,-1
     200     369    1746     369     6371743.151  688.44     700  1742.3
Permanent Ineff=
       F       F       F
Bank Sta=647.1,676.2
XS Rating Curve= 0 ,0
Exp/Cntr=0.5,0.3

Type RM Length L Ch R = 1 ,8812    ,120.1,112.6,102.9
XS GIS Cut Line= 4
2470531.31248272581514.2934604092470997.62228027581708.106013606
2471158.14131456  581926.9182162     2471375.316      582068.268
#Sta/Elev= 30
       0  1776.5      34 1762.88      60 1750.04    68.7 1747.61      86 1745.41
   198.6 1744.51   233.3 1742.56   263.6 1743.07   294.3 1740.87   332.9 1743.06
   397.8 1739.72   441.2 1740.96     565 1739.58   597.7 1740.64   605.1 1738.04
   610.8 1734.94   621.8 1734.31   635.4 1734.89   642.1 1738.01   648.9 1740.85
   672.1 1742.06   750.3 1740.96   770.6 1746.64   786.6  1748.8   811.5 1759.16
   824.8 1766.16   843.9 1768.48   858.2 1775.61   939.3 1806.48  1035.5 1833.33
#Mann= 12 ,-1 , 0
       0      .1       0  166.87     .12       0     243      .1       0
  400.53     .12       0  528.12    .055       0  570.99     .06       0
   605.1    .045       0   642.1     .06       0  680.88      .1       0
  746.48     .06       0  892.21      .1       0 1026.42     .12       0
#XS Ineff= 2 , 0
          596.68 1745.55  678.49         1746.56
Permanent Ineff=
       F       F
Bank Sta=605.1,642.1
XS Rating Curve= 0 ,0
Exp/Cntr=0.5,0.3

Type RM Length L Ch R = 1 ,8699    ,231.5,240.1,246.5
XS GIS Cut Line= 2
2470498.19659713581568.2868442942471283.09558125 582074.49510053
#Sta/Elev= 30
       0 1785.48    24.5 1775.13    86.3 1761.75   129.2 1747.67   167.2    1743
     191 1741.59   357.6 1738.45   400.5  1739.4   438.5 1738.89   473.9 1736.91
     514 1737.39   543.3 1735.17   557.5 1736.39   571.8 1734.12   586.1 1736.46
   589.7 1735.65   595.6 1733.02   600.4 1732.49   612.8 1732.99   619.4 1735.61
   628.9 1738.57   740.1 1737.57   771.7 1739.32   809.8 1760.85   824.1 1763.65
   833.6 1768.94   843.1 1770.66   852.6 1777.36   857.4 1779.56     934 1806.39
#Mann= 6 ,-1 , 0
       0      .1       0  112.91      .1       0   589.7    .045       0
   619.4      .1       0  704.92     .06       0  851.68      .1       0
#XS Ineff= 2 , 0
          555.05 1744.64  631.58         1745.32
Permanent Ineff=
       F       F
Bank Sta=589.7,619.4
XS Rating Curve= 0 ,0
Exp/Cntr=0.3,0.1

Type RM Length L Ch R = 1 ,8459    ,435.9,434.6,427
XS GIS Cut Line= 2
     2470591.347       581693.08     2471058.588      582372.485
#Sta/Elev= 30
       0 1758.44    26.5  1753.5    48.4 1747.39    97.8 1742.16   162.4 1738.68
   236.7 1738.13   325.9 1733.37   360.4  1733.4     376 1732.37   389.2 1732.97
   397.8 1729.91   400.7 1728.34   406.4 1727.24   420.8 1727.64   424.5 1728.65
   426.6 1730.26   429.5 1732.85   434.3 1734.47   452.5 1732.02   464.8 1733.33
   504.2 1732.49   542.5 1734.14   593.4 1733.12   656.7 1733.42   667.3 1735.57
   683.7 1741.49   706.1 1752.78   731.5 1763.27   783.3 1774.66   824.6 1789.16
#Mann= 8 ,-1 , 0
       0      .1       0   27.82      .1       0   42.43      .1       0
  258.89      .1       0   397.8    .045       0   426.6      .1       0
  583.57     .06       0  724.82      .1       0
#XS Ineff= 2 , 0
          392.18 1736.21  433.69         1736.52
Permanent Ineff=
       F       F
Bank Sta=397.8,426.6
XS Rating Curve= 0 ,0
Exp/Cntr=0.3,0.1

Type RM Length L Ch R = 1 ,8025    ,442.2,442.2,439.5
XS GIS Cut Line= 3
2470323.14154014582142.859590475     2470531.032      582335.571
 2470993.5768068582784.944857141
#Sta/Elev= 30
       0 1801.15    92.2 1791.32   127.1 1784.14   141.3 1777.78   152.6 1776.79
   195.8 1764.94   211.9 1758.88   235.4 1745.58   241.3 1740.72   253.1 1727.62
   258.9 1723.06   268.6 1722.12   277.1 1719.77   288.2 1719.43   308.2    1723
   311.2 1724.49   339.4 1728.71   385.8  1725.6   500.6 1728.13     604  1725.3
   623.3 1726.31   634.4 1729.03   656.2 1729.38   673.2 1738.65   695.8 1746.57
   734.8 1748.06   773.8 1752.89   827.8 1753.79     891 1786.35   928.4 1802.97
#Mann= 6 ,-1 , 0
       0      .1       0   268.6    .045       0   308.2      .1       0
  402.83     .05       0  575.62     .06       0  742.13      .1       0
#XS Ineff= 2 , 0
                          341.23         1739.35
Permanent Ineff=
       F       F
Bank Sta=268.6,308.2
XS Rating Curve= 0 ,0
Exp/Cntr=0.3,0.1

Type RM Length L Ch R = 1 ,7582    ,314.1,310.5,299.2
XS GIS Cut Line= 2
2470023.19233877582475.382590475 2470612.3804898582981.092496598
#Sta/Elev= 30
       0 1808.74    75.9 1793.92   115.4 1783.61   152.8 1767.38   173.4 1753.34
   183.9 1747.96   189.2 1743.56   195.1 1736.67   200.7 1732.76   212.1 1730.45
   226.5 1724.62   246.1 1721.89   254.6 1717.84   263.1 1715.06   273.5 1714.59
   285.8 1715.33   291.5 1717.88   299.9 1721.34   315.7 1719.08   331.5 1719.41
     342 1721.92   351.1  1722.3   637.6 1720.44   668.9 1718.99     690 1719.94
   700.5 1723.78   721.6    1725   732.1 1734.27   753.9  1748.3   776.5 1756.86
#Mann= 9 ,-1 , 0
       0     .12       0    4.21      .1       0   46.17     .12       0
  158.24      .1       0   174.5      .1       0   254.6    .045       0
   291.5      .1       0  431.14     .05       0  687.79     .06       0
#XS Ineff= 2 , 0
                          349.73         1730.79
Permanent Ineff=
       F       F
Bank Sta=254.6,291.5
XS Rating Curve= 0 ,0
Exp/Cntr=0.3,0.1

Type RM Length L Ch R = 1 ,7272    ,117.7,120.8,122.7
XS GIS Cut Line= 2
2469772.99781134582780.7166373392470564.81373469 583079.76141421
#Sta/Elev= 30
       0 1807.51    10.4 1803.46    23.2  1800.4   117.3 1784.76   151.5 1775.68
   232.8 1740.85   251.3 1729.25   254.1 1726.55   258.4 1719.63   262.7 1713.91
   266.5 1711.49   271.2 1711.24   282.4 1711.88   294.7 1714.68   309.7  1719.9
   322.7 1717.44   356.9 1714.91   395.2  1716.3   443.8 1716.53   524.5 1715.53
     597 1717.91   701.4 1719.11   710.7  1720.8   720.2 1725.12   737.3 1726.58
   741.6 1729.49   745.9 1733.89   750.1 1737.01   767.2 1745.35   846.4 1771.28
#Mann= 9 ,-1 , 0
       0      .1       0  115.26     .12       0  130.63      .1       0
   262.7    .045       0   294.7      .1       0  328.58      .1       0
  458.96     .05       0  688.09     .06       0  802.65      .1       0
#XS Ineff= 2 , 0
                          310.43         1724.61
Permanent Ineff=
       F       F
Bank Sta=262.7,294.7
XS Rating Curve= 0 ,0
Exp/Cntr=0.3,0.1

Type RM Length L Ch R = 1 ,7151    ,178.2,176.5,173.8
XS GIS Cut Line= 2
2469710.54697552582833.2267626952470433.41718433583217.952434687
#Sta/Elev= 30
       0 1797.46    83.6 1783.18    97.2 1780.69   110.8 1776.86   134.5  1765.7
     167  1742.1   190.5 1720.99   199.5 1716.25   213.2 1713.75   258.5 1715.68
   285.7 1715.76   301.5 1713.63   335.21711.813   349.1 1708.62   361.1 1712.15
   389.9 1722.25   406.5 1714.46   421.6 1712.21   462.4 1714.88   498.7 1712.86
   539.6 1715.88   648.2 1716.72   664.8 1720.46   679.9  1725.8   716.2 1728.35
   735.7 1739.91   756.9 1740.16   770.5 1746.79   781.1 1748.95   818.9 1753.92
#Mann= 11 ,-1 , 0
       0      .1       0    83.6     .12       0    97.2      .1       0
   213.2    .045       0   258.5      .1       0   301.5      .1       0
   335.2    .045       0   361.1      .1       0   421.6     .05       0
   664.8     .06       0   781.1      .1       0
#XS Ineff= 2 , 0
          288.34 1724.49  391.23         1729.12
Permanent Ineff=
       F       F
Bank Sta=335.2,361.1
XS Rating Curve= 0 ,0
Exp/Cntr(USF)=0,0
Exp/Cntr=0.3,0.1

Type RM Length L Ch R = 1 ,6975    ,374.7,378.9,379.5
XS GIS Cut Line= 3
     2469586.766      583018.699     2469971.874      583166.586
     2470343.635      583336.773
#Sta/Elev= 30
       0  1798.9    98.5 1764.41   158.5 1730.71   184.2 1709.78   231.4 1709.55
   248.5 1707.87   257.1 1710.81   299.9 1709.96   312.8  1711.5   329.9 1709.95
   351.3 1712.34   396.4 1710.55   402.7 1707.59   411.3 1706.17   420.1 1707.54
   424.5 1710.62   428.9 1712.47   466.2 1711.38   478.3 1709.58   496.4 1711.61
   534.5 1709.73   556.5 1712.54   582.9 1712.12   653.3 1716.16   672.7 1721.14
   689.5 1731.64   710.4 1733.69   719.7 1741.36   732.4 1746.07   821.4  1769.2
#Mann= 4 ,-1 , 0
       0      .1       0   396.4    .045       0   424.5      .1       0
  667.03     .06       0
Bank Sta=396.4,424.5
XS Rating Curve= 0 ,0
Exp/Cntr=0.3,0.1

Type RM Length L Ch R = 1 ,6596    ,367.7,366.5,360.7
XS GIS Cut Line= 2
2469367.93441878583250.3106800022470128.55510694583677.690290612
#Sta/Elev= 30
       0 1866.69    58.3 1831.62   146.4  1772.2   184.6 1748.01   237.2 1719.01
     251 1708.29   260.2 1703.25   333.6 1703.73   347.3 1700.95   388.6 1704.51
   411.6 1702.05     434 1702.53     449 1704.15   458.5 1702.92   469.6 1701.78
   478.4 1702.39   494.2 1700.79   540.1 1705.85   544.6 1707.58   560.6  1720.2
   566.5 1722.92   604.3 1724.15     641 1730.44   666.4 1738.64   703.4 1739.32
     734 1736.72   768.8 1738.78   786.8 1745.69   815.3 1754.07   872.5 1767.44
#Mann= 7 ,-1 , 0
       0      .1       0  100.15      .1       0   458.5    .045       0
   478.4      .1       0  558.71     .06       0  716.57      .1       0
  735.03      .1       0
Bank Sta=458.5,478.4
XS Rating Curve= 0 ,0
Exp/Cntr=0.3,0.1

Type RM Length L Ch R = 1 ,6229    ,298.2,309.7,318.6
XS GIS Cut Line= 2
2469154.33101134583641.3279854712470092.61794857583925.048179592
#Sta/Elev= 30
       0 1801.43    71.5 1754.32   113.3 1728.61   142.5 1708.59   159.2 1699.59
   165.2 1697.64   203.7 1695.42     293 1697.46   359.8 1697.35   376.5 1696.01
   415.5 1698.32   460.4 1696.61   472.6 1697.91   506.1 1697.39   518.6 1695.29
   531.4 1696.61     552 1697.83   572.9 1696.95   577.1 1698.14   610.5 1724.35
   630.5 1727.96   652.9 1738.34   673.2 1740.47   726.7 1740.73   756.8 1751.07
   790.2  1760.4   802.8 1761.76   862.2 1781.57   906.4 1794.37   980.2 1811.98
#Mann= 8 ,-1 , 0
       0      .1       0    59.9      .1       0  205.85      .1       0
  431.15      .1       0   506.1    .045       0   531.4      .1       0
  612.56     .06       0  723.09      .1       0
Bank Sta=506.1,531.4
XS Rating Curve= 0 ,0
Exp/Cntr=0.3,0.1

Type RM Length L Ch R = 1 ,5919    ,266.7,266.8,264.8
XS GIS Cut Line= 2
2469126.37223104583675.2542310412469839.27991921 584389.74775443
#Sta/Elev= 30
       0 1801.18    23.2 1786.94   106.8 1730.04   130.1 1718.13   147.8 1711.55
   170.4 1699.55   181.7 1695.49     295 1693.04   327.2 1694.04   342.2 1690.49
   372.4 1692.65   432.8 1692.35   445.9 1693.88   502.4 1692.75   526.1 1690.28
   532.9 1691.07   540.2 1694.07   551.6 1695.58   566.8 1692.23   612.1 1692.68
   639.2 1690.91     659 1692.91   691.4 1696.02   714.1 1706.22   735.4 1713.01
   777.8 1712.62   801.9 1706.61   841.4 1711.56   923.6 1742.59  1009.3 1769.96
#Mann= 6 ,-1 , 0
       0      .1       0  194.84      .1       0   502.4    .045       0
   540.2      .1       0     659     .06       0  829.08      .1       0
Bank Sta=502.4,540.2
XS Rating Curve= 0 ,0
Exp/Cntr=0.3,0.1

Type RM Length L Ch R = 1 ,5653    ,334,328.6,317.3
XS GIS Cut Line= 3
2468846.52128664583879.4919074992469058.40922498583992.935885808
2469730.18608336584633.562647505
#Sta/Elev= 30
       0  1831.8    63.8 1802.71   127.3 1770.24   150.4 1761.59   182.9 1754.39
   266.4 1742.01   312.7  1733.5   351.4 1722.41   406.6 1690.44   450.8 1686.22
   471.1 1688.62   505.1 1688.48   521.4 1686.63   539.3 1689.14   553.2 1689.11
     562 1686.85   573.6 1686.45   594.6  1689.3   605.6 1693.03   637.3 1686.47
     672 1689.71   841.8 1689.42   904.1    1691   915.3 1694.12   943.6 1708.62
   964.9 1711.29   975.9 1718.52  1069.9 1755.85  1124.2 1772.75  1168.6 1780.74
#Mann= 8 ,-1 , 0
       0      .1       0  250.52      .1       0  425.09      .1       0
   553.2    .045       0   594.6      .1       0  794.06     .05       0
  908.36     .06       0 1072.81      .1       0
Bank Sta=553.2,594.6
XS Rating Curve= 0 ,0
Exp/Cntr=0.3,0.1

Type RM Length L Ch R = 1 ,5324    ,410.3,416.9,417.6
XS GIS Cut Line= 2
2468809.03848393584328.6231831732469747.17373478584674.763844004
#Sta/Elev= 30
       0 1785.28    40.2 1762.55    65.8 1749.52    78.6 1745.42   138.3 1732.87
     190 1717.32   202.2 1709.25   224.2 1688.92   230.4 1684.74   244.8 1682.45
   264.7 1683.47   313.1 1683.33   342.9 1687.72   368.5 1682.84   419.7 1682.95
   436.7 1685.46   509.2 1685.39   556.1 1682.65   590.2 1686.02   675.5 1685.97
   722.4 1688.42   730.9 1690.64   742.3 1695.58   760.7 1707.51   777.8 1708.75
   781.7 1710.11   794.8 1718.82   884.4 1757.15   935.5 1772.76    1000 1784.02
#Mann= 8 ,-1 , 0
       0      .1       0  123.35      .1       0   230.4    .045       0
   264.7      .1       0  579.62     .05       0  693.69      .1       0
  701.02     .06       0  901.69      .1       0
Bank Sta=230.4,264.7
XS Rating Curve= 0 ,0
Exp/Cntr=0.3,0.1

Type RM Length L Ch R = 1 ,4907    ,258.2,253.3,247.6
XS GIS Cut Line= 2
2468628.63412151584635.4675320112469472.79720852585115.126376015
#Sta/Elev= 30
       0 1802.63    33.4 1797.48      53  1792.6    68.6 1786.88   118.5 1764.13
   140.4 1752.85   209.3 1709.08   250.9 1688.99   265.2 1679.61   269.3 1677.96
   283.1 1678.89   301.5 1677.06     318 1678.76   324.5 1680.66   370.5 1678.67
     403 1679.25   470.5 1677.47   513.1 1679.41   617.2 1675.81   719.9  1680.5
   733.9 1686.53   752.1  1700.2   756.9 1702.62   779.9 1704.85   798.3 1717.03
   830.5 1725.63   863.6 1739.94   904.7 1746.24   946.2 1748.14   970.9  1752.4
#Mann= 8 ,-1 , 0
       0     .05       0  174.48      .1       0   283.1    .045       0
     318      .1       0  429.41     .05       0  732.48    .055       0
  811.81     .06       0  889.38      .1       0
Bank Sta=283.1,318
XS Rating Curve= 0 ,0
Exp/Cntr=0.3,0.1

Type RM Length L Ch R = 1 ,4654    ,353.3,356.3,358.3
XS GIS Cut Line= 2
2468524.96595976584905.1016937562469506.78657304 585234.39203449
#Sta/Elev= 30
       0  1791.6    69.4 1777.96    94.7 1769.24   115.8 1759.04     145  1742.8
   211.3 1701.79   233.9 1691.52     265  1686.3   305.6 1676.95   326.7 1675.22
   352.1 1675.15   360.5 1677.67   373.1 1675.16     390 1676.98   415.3 1675.69
   558.9 1674.06   584.3    1675     601  1683.8     660 1704.68   672.6 1705.05
   682.1 1708.89     698 1708.82   710.5 1715.39   723.3 1717.74   803.5 1728.03
   816.1 1732.09   879.4  1747.2   938.5 1757.76   963.3 1763.52  1035.6 1785.27
#Mann= 8 ,-1 , 0
       0      .1       0   93.57      .1       0   326.7    .045       0
   352.1      .1       0  542.47     .05       0  654.69    .055       0
   657.6     .06       0  766.91      .1       0
Bank Sta=326.7,352.1
XS Rating Curve= 0 ,0
Exp/Cntr=0.3,0.1

Type RM Length L Ch R = 1 ,4298    ,267.8,269.7,412.3
XS GIS Cut Line= 2
2468450.92892527585201.1717742332469315.90534727585475.476254509
#Sta/Elev= 30
       0 1776.66     8.2 1770.79    20.8 1767.24    45.8 1749.78    90.4 1720.81
   131.8 1696.24   146.7 1691.45   180.2  1674.4   188.6 1670.46   214.7 1671.26
   243.2 1672.26   285.2  1670.5   306.1 1671.38   314.5  1670.2   336.5 1672.72
   360.7 1673.58   532.7 1671.04   587.3 1671.44   595.7 1672.42   600.2 1674.43
   612.5 1692.84   637.6 1706.53   657.5 1707.88   676.6 1712.31   702.1 1716.25
   746.7 1726.53   756.3 1727.64   772.2 1734.38   848.7 1762.19   907.4 1782.13
#Mann= 10 ,-1 , 0
       0      .1       0   47.42      .1       0  116.48      .1       0
   180.2    .045       0   214.7      .1       0   266.6      .1       0
  485.77    .025       0  561.57     .06       0  672.84    .055       0
  704.95      .1       0
Bank Sta=180.2,214.7
XS Rating Curve= 0 ,0
Exp/Cntr=0.3,0.1

Type RM Length L Ch R = 1 ,4028    ,283.3,326.6,434.1
XS GIS Cut Line= 3
2468360.80182676585384.5251230712468465.49770437585514.281499086
2469225.60074785585542.907928928
#Sta/Elev= 30
       0 1745.33     156 1729.16     180 1724.72     216  1712.5     256 1695.68
   288.1  1683.6   296.1 1679.65   304.1 1672.68   307.4 1670.75   312.1 1669.59
   320.1 1669.34   664.3 1669.34   668.3 1671.59   692.3 1685.39   727.9 1698.32
   740.4  1704.3   752.4 1711.23   756.4 1711.89   768.4 1711.85   772.4 1713.94
   776.4 1717.27   780.4 1719.37   796.4 1720.34   800.4 1722.55   808.4 1728.27
   816.4  1731.7   832.4    1737   848.5 1741.48   893.7 1757.33   927.4 1767.18
#Mann= 8 ,-1 , 0
       0      .1       0    56.4     .12       0  207.91      .1       0
   307.4    .045       0   668.3    .025       0  714.43     .06       0
  815.73      .1       0  917.04      .1       0
Bank Sta=307.4,668.3
XS Rating Curve= 0 ,0
Exp/Cntr=0.3,0.1

Type RM Length L Ch R = 1 ,3701    ,239.5,348.9,493.2
XS GIS Cut Line= 3
2468354.37238751585422.4629783082468252.56933256585661.917440622
2469054.79983251586047.712493337
#Sta/Elev= 30
       0  1742.3    12.2 1739.52    30.9  1732.4    39.9 1730.91   216.6 1725.11
   271.3 1721.69   284.8 1719.06   324.7 1707.04   355.8 1699.56   391.4 1697.22
   445.4 1695.75   457.9 1694.61   472.4 1687.23   493.3 1670.83   497.9  1669.7
   506.7 1669.34     904 1669.34   912.6 1670.17   932.8 1680.96   963.9 1693.47
   981.9 1701.88  1030.5 1726.36  1038.8 1730.99  1057.1 1743.58  1083.8 1745.88
  1104.8 1749.99  1116.7 1755.43  1122.7 1756.92  1134.9 1757.77  1150.4  1756.4
#Mann= 12 ,-1 , 0
       0      .1       0   14.49     .05       0  118.57     .12       0
  129.32     .05       0  244.15     .12       0  352.31      .1       0
  408.28    .055       0   493.3    .045       0   912.6      .1       0
  924.72    .055       0  957.73     .06       0 1096.87      .1       0
Bank Sta=493.3,912.6
XS Rating Curve= 0 ,0
Exp/Cntr=0.3,0.1

Type RM Length L Ch R = 1 ,3352    ,245.9,414.6,266.1
XS GIS Cut Line= 3
2468313.00770002585436.0834329072468185.29400477585679.611952422
 2468588.6003511586509.402384524
#Sta/Elev= 30
       0 1735.12     7.7  1732.2    21.2 1730.85    84.5 1730.63   156.7 1727.32
   256.1 1724.31   296.4 1721.75   309.8 1717.47   323.1 1717.08   327.6 1716.06
   380.9  1696.3   407.2 1693.52   541.9 1687.14   554.4 1683.86   571.1 1677.78
   585.5 1670.17   594.4 1669.34   901.3 1669.99   909.7 1674.39   945.7 1698.64
   994.7 1727.97  1032.7  1746.8  1066.4 1762.07  1079.2 1769.42    1097 1771.13
  1110.5 1779.06  1126.9 1784.58  1143.4 1788.72  1163.7 1791.66  1197.6 1793.54
#Mann= 11 ,-1 , 0
       0      .1       0    6.46     .05       0   33.74     .12       0
  127.79     .05       0  249.12      .1       0  457.31    .025       0
   585.5    .045       0   901.3     .05       0   967.5      .1       0
 1069.53     .06       0 1171.57     .05       0
Bank Sta=585.5,901.3
XS Rating Curve= 0 ,0
Exp/Cntr=0.3,0.1

Type RM Length L Ch R = 1 ,2938    ,336.9,270.6,711.6
XS GIS Cut Line= 3
2468286.30617365  585419.32130042468041.46904762585977.051520841
2468347.35190425586616.415303846
#Sta/Elev= 30
       0 1739.85      17 1733.32    34.5 1731.84   196.1 1727.24   293.8 1723.19
   305.3  1721.7   331.5 1721.63   353.4 1717.92   406.1 1703.98   442.81697.247
     564 1689.03   576.1 1689.03   593.6 1691.48   609.1 1691.25   628.9 1688.23
   651.1 1681.93   726.4 1669.86   741.8 1669.34  1050.1 1669.34  1055.3 1669.57
  1060.9 1671.33  1085.6 1687.02  1121.8 1707.44  1165.4 1728.41    1192 1739.99
  1218.6 1750.26  1260.9 1764.01  1280.3 1774.57  1297.9 1777.68  1317.9 1777.97
#Mann= 8 ,-1 , 0
       0      .1       0   32.41     .12       0  154.65     .05       0
   276.9      .1       0  320.95     .05       0   442.8    .045       0
  1060.9      .1       0 1137.37    .055       0
Bank Sta=442.8,1060.9
XS Rating Curve= 0 ,0
Exp/Cntr=0.3,0.1

Type RM Length L Ch R = 1 ,2667    ,116.3,102,94.9
XS GIS Cut Line= 2
2467764.28296039585654.3008738052468115.85258465586619.880723102
#Sta/Elev= 30
       0 1759.48    27.3 1748.93    47.5  1743.1      56 1739.86    85.8 1725.89
    98.5 1719.07   105.4 1716.26   111.3 1714.93   119.8 1714.49   167.8 1714.17
     239 1714.52   264.5 1715.09   273.1 1716.77   302.9 1726.77   311.3 1728.65
   315.6 1728.97   339.4 1728.23   451.5 1729.92   526.7 1729.78     697 1730.53
     849 1730.38   941.4 1728.99   945.7 1729.69   949.9 1731.74   962.7 1739.03
   971.2 1745.02   975.5 1746.89     984 1748.65  1005.3 1759.78  1027.6 1769.12
#Mann= 8 ,-1 , 0
       0     .05       0   70.16      .1       0   111.3    .045       0
   264.5     .05       0  467.81    .025       0  666.66     .05       0
  766.07    .055       0   964.9     .05       0
Bank Sta=111.3,264.5
XS Rating Curve= 0 ,0
Exp/Cntr=0.3,0.1

Type RM Length L Ch R = 1 ,2414    ,100.4,66.7,48.2
XS GIS Cut Line= 3
2467473.05040176585845.2127732232467722.72630587586089.076326897
2467825.11982214586646.899482304
#Sta/Elev= 30
       0 1778.43    13.9 1777.82    25.3 1773.71      94 1736.75   126.8 1721.91
   135.3 1713.45   142.2 1710.68   296.6 1710.32   324.8 1719.15   334.4 1720.35
   345.9 1719.08     411 1691.43   444.4  1681.9   464.7 1678.47   509.5 1666.57
   517.6 1663.67   537.9  1653.8     598 1651.19   643.7 1644.76   680.3 1645.46
   700.6  1647.7   704.7 1649.17     725 1665.79   781.9 1703.27   802.3 1715.32
   838.9 1733.64     847 1738.67   863.3 1745.78   891.7 1756.92   916.2 1764.93
#Mann= 8 ,-1 , 0
       0      .1       0   27.99      .1       0   142.2    .045       0
   296.6     .05       0  384.72      .1       0  677.42    .055       0
  774.99      .1       0  872.55    .055       0
#XS Ineff= 2 , 0
                          331.58         1733.52
Permanent Ineff=
       F       F
Bank Sta=142.2,296.6
XS Rating Curve= 0 ,0
Exp/Cntr=0.3,0.1

Type RM Length L Ch R = 1 ,2347    ,91,69.5,56
XS GIS Cut Line= 3
2467397.95886775 585965.641258352467705.50452938586113.317369002
2467775.95551795586628.151516232
#Sta/Elev= 30
       0  1771.2    45.2 1745.91    71.9 1732.55    85.2 1727.96   104.5 1726.34
   107.4 1724.54   118.4 1712.09   125.1 1708.61   277.3 1708.61   292.3  1713.5
   302.6 1713.68   320.4 1707.48   341.2 1704.88   362.9 1697.22   444.5 1681.27
   459.8  1675.3   492.1 1655.21     507 1650.54   516.4 1648.86   532.5 1648.72
   576.9 1641.31   601.1 1644.08   641.5 1644.74   657.7 1646.48   663.3 1649.72
   670.4 1659.29   677.8 1665.74   758.6  1710.3   794.9 1726.85   860.8  1748.3
#Mann= 6 ,-1 , 0
       0      .1       0   21.99      .1       0   125.1    .045       0
   277.3     .05       0  355.55      .1       0  745.74      .1       0
#XS Ineff= 2 , 0
                          294.74         1728.68
Permanent Ineff=
       F       F
Bank Sta=125.1,277.3
XS Rating Curve= 0 ,0
Exp/Cntr(USF)=0,0
Exp/Cntr=0.3,0.1

Type RM Length L Ch R = 1 ,2278    ,70.3,40.8,33.8
XS GIS Cut Line= 3
 2467376.2816405586080.8015281252467696.02074246586153.962170099
2467756.98794411586615.958075903
#Sta/Elev= 30
       0 1762.11    45.2 1737.69    63.2 1729.39    80.6 1722.98    92.8 1716.04
     101  1709.3   109.2 1706.92   254.2 1706.39   265.1 1708.39   269.2 1708.11
     341  1693.3   384.7 1686.46   393.5  1682.7   413.7 1670.57   421.7 1664.71
   441.9 1653.16   462.1  1647.9   486.3 1646.31   506.5 1639.15   525.8 1638.55
   546.8 1639.14   562.9 1643.72   591.2 1644.37   603.3 1646.22   611.4 1650.49
   631.5 1669.68   693.1 1702.71   724.3 1717.31   756.6    1729     794 1740.16
#Mann= 6 ,-1 , 0
       0      .1       0   15.57      .1       0   109.2    .045       0
   254.2     .05       0  401.23      .1       0   693.9      .1       0
#XS Ineff= 2 , 0
                          266.67         1724.28
Permanent Ineff=
       F       F
Bank Sta=109.2,254.2
XS Rating Curve= 0 ,0
Exp/Cntr(USF)=0,0
Exp/Cntr=0.3,0.1

Type RM Length L Ch R = 1 ,2237    ,31.9,20.3,19
XS GIS Cut Line= 3
2467358.38431405586142.2070111342467692.90942596586179.376468013
2467749.69609619586620.247525993
#Sta/Elev= 30
       0 1764.76    12.4 1761.04    28.5  1752.2    64.8 1734.79      97 1722.75
   117.1 1707.96   121.1  1706.2   169.4 1705.87   258.81703.793   306.2 1699.75
   336.6 1693.36   364.3 1688.87   368.4 1687.68   384.5 1679.36   424.8 1653.38
     445 1647.87   469.2 1646.21   485.3 1639.04   505.5 1638.45   533.7 1638.73
   537.7 1639.24   549.8  1643.7     574  1644.2   586.1 1646.16   594.2 1650.27
   606.3 1662.31   618.4 1671.66   662.9 1695.64   715.2 1718.49   781.1 1739.27
#Mann= 7 ,-1 , 0
       0      .1       0   43.51      .1       0   146.6      .1       0
   169.4    .045       0   258.8     .05       0  385.17      .1       0
  677.86      .1       0
#XS Ineff= 2 , 0
                          260.91         1732.61
Permanent Ineff=
       F       F
Bank Sta=169.4,258.8
XS Rating Curve= 0 ,0
Exp/Cntr(USF)=0,0
Exp/Cntr=0.3,0.1

Type RM Length L Ch R = 1 ,2216    ,399.9,408.6,425.2
XS GIS Cut Line= 3
2467334.18343614586164.570405239 2467687.9051194586196.437223551
2467741.44137416586629.825952591
#Sta/Elev= 30
       0 1758.83    33.4 1757.78    44.7  1755.2    92.9 1733.47     121 1724.89
   129.1 1719.96   145.1 1707.82   149.2  1705.9   189.3 1704.91   216.3  1702.8
   279.71700.415   329.1  1697.4   369.7 1689.66   381.8 1683.96   422.1 1657.48
   431.6 1652.39   450.3 1647.21   474.3 1645.52   486.6 1639.12   499.8 1638.59
     539 1638.71   551.1 1643.17   575.3    1644   587.4 1646.23   596.7 1652.46
   611.5    1665   623.6  1673.1     676 1699.93     733 1721.76   791.8 1739.17
#Mann= 7 ,-1 , 0
       0      .1       0   71.62      .1       0  174.14      .1       0
   216.3    .045       0   279.7     .05       0  387.65      .1       0
  680.38      .1       0
#XS Ineff= 2 , 0
                          280.15         1723.73
Permanent Ineff=
       F       F
Bank Sta=216.3,279.7
XS Rating Curve= 0 ,0
Exp/Cntr(USF)=0,0
Exp/Cntr=0.3,0.1

Type RM Length L Ch R = 1 ,1808    ,290.6,290.4,289.9
XS GIS Cut Line= 2
2467269.14916198 586269.470984122467665.19904356586731.838399274
#Sta/Elev= 30
       0  1721.2    24.8  1706.3      44 1693.89    49.3 1688.59    54.5 1682.34
    59.8 1677.35    80.9 1660.02    86.1  1654.5    96.7 1640.17   101.9 1637.18
   112.5 1637.97   128.3  1637.4   246.1 1638.07   263.1 1638.49   285.8 1640.28
   292.1 1639.08   297.2 1637.04   302.1 1636.34   308.5 1636.83   314.2 1638.84
   323.1 1642.95   346.8 1644.93   365.3 1651.91   377.5 1659.09   381.1 1660.58
   436.2 1672.18   463.6 1680.65   524.1  1706.4   568.1 1723.54   608.8 1737.91
#Mann= 6 ,-1 , 0
       0      .1       0    28.9      .1       0   98.07      .1       0
   292.1    .045       0   314.2      .1       0  479.62      .1       0
Bank Sta=292.1,314.2
XS Rating Curve= 0 ,0
Exp/Cntr=0.3,0.1

Type RM Length L Ch R = 1 ,1517    ,266.6,249,233.6
XS GIS Cut Line= 2
2467034.01530426586449.9240159062467415.97929868586878.115280388
#Sta/Elev= 30
       0 1712.85    40.9 1704.54    46.5 1702.69    57.9 1697.04    74.9 1687.84
   103.2 1669.25   115.3 1659.58   124.6 1649.42   131.5 1643.66     146 1637.33
   151.3 1636.25   181.4 1634.29   307.2 1636.15   315.7  1635.9   319.6 1635.02
   325.6    1633   331.6 1632.67   337.6 1633.48   341.2  1634.9   346.8  1636.1
   358.2 1636.25   366.7 1638.09   385.7 1647.63   403.3  1659.6   408.7 1661.18
   499.8 1668.65   511.9 1670.23   542.7 1675.86   559.3 1681.07   573.8  1687.3
#Mann= 7 ,-1 , 0
       0      .1       0   26.21      .1       0   92.19      .1       0
   319.6    .045       0   341.2      .1       0  395.65      .1       0
   440.7      .1       0
#XS Ineff= 2 , 0
                          350.58          1638.6
Permanent Ineff=
       F       F
Bank Sta=319.6,341.2
XS Rating Curve= 0 ,0
Exp/Cntr=0.3,0.1

Type RM Length L Ch R = 1 ,1268    ,76.9,71.9,67.8
XS GIS Cut Line= 3
2466842.55255353586735.5616882822466957.94370325586874.411478322
2467270.64103862586897.489708264
#Sta/Elev= 30
       0 1696.48    12.8 1692.67    22.4 1687.51    42.3 1672.54    67.8 1652.05
    79.2 1640.06    82.3 1637.67    96.2 1637.49   108.3 1634.51     138 1631.65
   222.8 1631.37   285.6 1633.28   293.6 1632.49   301.7 1630.03   321.7 1628.64
   329.7 1628.84   336.8 1630.64   345.8 1632.41   365.8  1632.2   379.7 1634.19
   383.4 1635.53   397.9 1644.06   401.9  1645.4   417.1 1646.16   420.8 1647.08
     434 1655.02     438 1656.23   462.1 1661.44   478.1 1663.31   494.1 1666.37
#Mann= 3 ,-1 , 0
       0      .1       0   301.7    .045       0   336.8      .1       0
#XS Ineff= 2 ,-1
       0  284.35 1636.43     353494.0869 1636.43
Permanent Ineff=
       F       F
Bank Sta=301.7,336.8
XS Rating Curve= 0 ,0
Exp/Cntr(USF)=0,0
Exp/Cntr=0.5,0.3

Type RM Length L Ch R = 1 ,1197    ,57.1,48.5,44.3
XS GIS Cut Line= 4
2466799.40257681586758.6782806622466976.49970785586989.147149829
2467177.25022284 586915.761009912467312.49905922586990.966640901
#Sta/Elev= 30
       0  1695.8    20.4 1692.46    45.3 1681.02    62.4 1675.54    73.8 1669.17
    85.3  1661.2    99.5 1644.66   102.4 1643.59   116.6 1644.22   130.2 1636.62
   141.5 1633.07     163 1631.69   182.2 1633.05   216.5 1631.35   257.5 1631.52
     293 1629.71   382.5 1630.66   386.7 1629.79   395.3 1627.63   406.4  1629.5
   467.7 1634.36   480.4 1637.17   497.5 1643.95   515.3 1645.24   519.6 1647.25
   528.4 1653.93   535.5 1656.54   593.1 1670.71     616 1677.48   659.1  1692.4
#Mann= 3 ,-1 , 0
       0      .1       0   386.7    .045       0   406.4      .1       0
#XS Ineff= 3 ,-1
     120     182    1635     182     386    1630     407     500  1630.5
Permanent Ineff=
       F       F       F
Bank Sta=386.7,406.4
XS Rating Curve= 0 ,0
Exp/Cntr(USF)=0,0
Exp/Cntr=0.5,0.3

Type RM Length L Ch R = 1 ,1148    ,93.6,128.2,157.5
XS GIS Cut Line= 4
2466779.68059293586766.4543558182466979.12003579587033.038684448
2467191.39399423586953.5875742872467313.52478924587028.679415336
#Sta/Elev= 30
       0 1695.69    20.5 1692.17    36.8 1685.16    56.8 1678.26    65.5 1673.58
    82.5 1669.49    91.1 1666.07   100.5 1660.19   110.4 1647.92   128.2  1648.2
     132 1646.82   142.5 1639.83   148.2 1637.43   171.1 1632.52   185.4 1631.22
   245.5 1630.81   330.2 1628.74   392.3 1630.19   405.1 1629.24     418 1626.95
     435 1627.08   446.2 1629.16   464.9 1632.65   503.4 1642.42   537.5 1643.68
   554.6 1654.14   572.9 1660.52   615.2 1672.98   680.9 1697.21     703 1704.38
#Mann= 5 ,-1 , 0
       0      .1       0   219.4    .055       0  252.99      .1       0
   405.1    .045       0   446.2      .1       0
Bank Sta=405.1,446.2
XS Rating Curve= 0 ,0
Exp/Cntr=0.5,0.3

Type RM Length L Ch R = 1 ,1020    ,81.1,82.6,82.5
XS GIS Cut Line= 3
2466724.98475003586731.6945356582467108.28999863587260.106415765
2467284.09720236587331.789083324
#Sta/Elev= 30
       0 1695.14    50.7 1693.13    78.1 1689.12   112.7 1680.98   146.1 1665.66
   157.1 1661.89   172.5 1651.68   195.4 1652.06   221.2 1638.47   241.4 1632.29
   280.7 1630.14   387.3 1628.53   418.8 1628.98   428.9 1631.34   438.9 1628.22
   463.5 1625.28   481.8  1628.3   496.2 1634.43   513.9 1636.19   533.4 1650.89
   562.3 1666.34   627.9 1695.14   643.4 1704.16   681.4 1702.03   702.8 1717.56
   711.6 1721.65   754.8 1730.92   776.4 1733.41     811 1732.56   842.7 1727.02
#Mann= 8 ,-1 , 0
       0      .1       0  265.75    .055       0  367.96      .1       0
   438.9    .045       0   481.8      .1       0  594.51     .06       0
  735.32    .055       0  741.42     .06       0
Bank Sta=438.9,481.8
XS Rating Curve= 0 ,0
Exp/Cntr=0.5,0.3

Type RM Length L Ch R = 1 ,937     ,138.3,139.1,140.8
XS GIS Cut Line= 4
2466701.57056694586729.0966199442466750.15145613586873.735176393
2467041.63679126587317.5878457992467266.87545932587479.892180134
#Sta/Elev= 30
       0 1683.01    28.8 1677.46   147.6 1663.33   182.7 1658.54   206.6 1649.59
   240.1 1642.65     264 1634.98   283.2 1631.61   312.7 1630.64   364.5 1628.94
   410.9 1630.49   460.2 1628.76   474.3 1630.65   483.1 1627.63   498.5  1624.3
   516.2 1627.81   525.3 1630.69   532.2 1629.64   541.6 1632.58   555.3 1632.78
   566.9 1632.47   581.3 1641.53     599 1652.36   632.5 1666.32   661.2  1672.8
   683.6 1673.72     749 1676.64   822.7 1678.78   891.1 1677.97   961.2 1668.44
#Mann= 12 ,-1 , 0
       0      .1       0   147.6     .06       0   312.7    .055       0
   364.5     .06       0   483.1    .045       0   516.2     .01       0
   555.3      .1       0   581.3    .055       0   683.6     .06       0
     749    .055       0   822.7     .06       0   891.1    .055       0
#XS Ineff= 2 , 0
          473.39  1635.8  525.42          1636.5
Permanent Ineff=
       F       F
Bank Sta=483.1,516.2
XS Rating Curve= 0 ,0
Exp/Cntr(USF)=0,0
Exp/Cntr=0.5,0.3

Type RM Length L Ch R = 1 ,798     ,93.5,90.2,84.9
XS GIS Cut Line= 4
2466689.59081827586711.0169981222466669.47350195 586921.41498191
2466931.91973304587421.1753455762467261.75631148587549.071161705
#Sta/Elev= 30
       0 1683.91     7.9 1683.33    28.2 1681.75    40.1 1677.96    56.1 1664.47
    72.2 1656.03    92.3 1638.58   100.3 1635.14   144.5 1635.44   184.7 1630.32
   272.6 1631.62   375.7 1631.59   480.8 1628.58   511.2 1625.79   558.2 1629.63
   583.5  1628.3   589.6    1626   609.8 1622.77     621 1625.54   646.8 1631.05
   687.3 1626.51   730.3 1627.86   859.7 1625.88   941.9 1626.58   959.1  1628.5
   993.4 1638.06  1044.9 1649.97  1090.4 1650.33  1110.1  1653.7  1129.6 1652.87
#Mann= 12 ,-1 , 0
       0      .1       0     7.9     .06       0   272.6      .1       0
   375.7     .06       0   480.8      .1       0   583.5     .06       0
   589.6    .045       0     621     .06       0   687.3    .055       0
   859.7     .06       0   993.4    .035       0  1090.4    .055       0
#XS Ineff= 2 , 0
          565.98 1632.77  645.21         1633.84
Permanent Ineff=
       F       F
Bank Sta=589.6,621
XS Rating Curve= 0 ,0
Exp/Cntr(USF)=0,0
Exp/Cntr=0.5,0.3

Type RM Length L Ch R = 1 ,708     ,298.2,299.5,299.6
XS GIS Cut Line= 4
2466671.07958173586689.1400822052466617.22871178 587086.29024808
2466977.35640456 587584.410795112467408.16336416 587613.01906977
#Sta/Elev= 30
       0 1687.99       9 1686.58    38.1  1673.7    54.2 1662.28    62.3 1649.93
    82.5 1635.53    87.2 1634.19     139 1634.92   179.6 1629.91   219.7 1629.81
   239.9 1631.61   400.8 1628.62   462.5 1629.68   613.8 1628.48     673 1625.45
   685.9 1628.28   696.9 1627.46   708.8 1623.41   722.4 1621.46   731.7 1623.39
   740.3  1625.8   786.5 1624.68   857.8 1627.17  1015.5 1623.86  1120.6 1625.37
  1289.4 1621.39  1333.5 1624.46  1385.7 1642.18  1432.6 1644.49  1447.2 1648.29
#Mann= 11 ,-1 , 0
       0     .06       0  295.12      .1       0  690.75     .06       0
   708.8    .045       0   731.7    .055       0  838.98     .05       0
  912.12    .055       0 1069.81    .035       0 1188.72     .02       0
 1273.67     .05       0  1375.6     .06       0
#XS Ineff= 2 , 0
                          742.28         1628.96
Permanent Ineff=
       F       F
Bank Sta=708.8,731.7
XS Rating Curve= 0 ,0
Exp/Cntr(USF)=0,0
Exp/Cntr=0.3,0.1

Type RM Length L Ch R = 1 ,409     ,193.9,192.3,163.2
XS GIS Cut Line= 4
2466641.57102246 586691.111474652466540.00045157587466.741288732
2466685.43104171587695.2750732382467585.81395315587718.627322023
#Sta/Elev= 30
       0 1670.46     7.8 1666.55    32.1 1645.01    48.7 1634.38    96.6 1634.67
   116.8 1631.44   165.2 1629.49   209.6 1630.25   341.2 1629.82   423.2 1621.91
   817.2 1620.03   842.3  1622.4   868.4  1619.7     882 1617.11   891.3 1619.44
   908.9 1624.24   919.9 1622.58   956.3 1621.09  1024.8 1620.43  1223.3 1621.62
  1317.8 1622.63  1422.6 1622.36  1457.5 1622.33  1522.6 1621.36  1622.6 1621.16
  1726.7  1620.3  1878.7 1620.05  1902.7 1624.87  1923.8 1635.54  1953.8 1642.31
#Mann= 15 ,-1 , 0
       0     .06       0   209.6      .1       0   868.4    .045       0
   891.3      .1       0   919.9     .06       0   956.3    .055       0
  1024.8     .05       0  1223.3    .055       0  1317.8    .035       0
  1422.6     .02       0  1457.5    .035       0  1522.6     .02       0
  1622.6    .055       0  1726.7     .05       0  1923.8     .06       0
#XS Ineff= 2 , 0
          841.16 1625.62   910.2         1626.11
Permanent Ineff=
       F       F
Bank Sta=868.4,891.3
XS Rating Curve= 0 ,0
Exp/Cntr(USF)=0,0
Exp/Cntr=0.3,0.1

Type RM Length L Ch R = 1 ,216     ,,,
XS GIS Cut Line= 4
2466637.45272817586657.7000266792466372.95363504587538.851075311
2466778.92898729587963.279852663 2467921.5035582587821.803593545
#Sta/Elev= 30
       0 1679.39    26.3 1668.08    35.3 1659.87    54.5 1637.48    59.7 1634.29
   105.7 1633.82     122 1629.26   134.8 1628.62   293.6 1630.28   360.4 1623.33
   520.3 1623.67   590.1 1617.04   627.7 1620.01   744.6 1617.92   840.7 1619.86
   934.2 1618.08     992 1619.19    1006 1616.23  1026.7 1615.21  1071.2 1616.18
  1080.6 1617.86    1183 1620.24  1356.6 1618.54  1382.4 1618.64    1620 1617.22
  1906.9 1620.94    2551 1616.84  2591.4 1618.36  2615.3 1623.95  2658.6 1634.61
#Mann= 9 ,-1 , 0
       0     .06       0   134.8      .1       0    1006    .045       0
  1071.2      .1       0    1183     .06       0  1356.6     .05       0
  1382.4      .1       0    1620     .05       0  2615.3     .06       0
#XS Ineff= 2 , 0
          990.59 1621.39 1175.75         1621.57
Permanent Ineff=
       F       F
Bank Sta=1006,1071.2
XS Rating Curve= 0 ,0
Exp/Cntr(USF)=0,0
Exp/Cntr=0.3,0.1
LCMann Table=0

Chan Stop Cuts=-1
Use User Specified Reach Order=0
Composite Channel Slope=5
